--- smsfrk.prj (project) ---

Proj Title=smsfrk
Current Plan=p01
Default Exp/Contr=0,0
English Units
Geom File=g01
Flow File=f01
Plan File=p01
BEGIN DESCRIPTION:
END DESCRIPTION:
DSS File=dss
DSS Export Rating Curves= 0
DSS Export Rating Curve Sorted= 0
DSS Export Volume Flow Curves= 0
DXF OffsetX= 0
DXF OffsetY= 0
DXF ScaleX= 0
DXF ScaleY= 0

--- smsfrk.p01 (plan) ---

Plan Title=Approximate Study - 100yr
Program Version=4.00
Short Identifier=Approximate
Geom File=g01
Flow File=f01
Subcritical Flow
K Sum by GR= 0
Std Step Tol= 0.01
Critical Tol= 0.01
Num of Std Step Trials= 20
Max Error Tol= 0.3
Flow Tol Ratio= 0.001
Split Flow NTrial= 30
Split Flow Tol= 0.02
Split Flow Ratio= 0.02
Log Output Level= 0
Friction Slope Method= 1
Unsteady Friction Slope Method= 2
Unsteady Bridges Friction Slope Method= 1
Parabolic Critical Depth
Global Vel Dist= 0 , 0 , 0
Global Log Level= 0
CheckData=True
Encroach Param=-1 ,0,0, 0
Run HTab= 0
Run UNet= 0
Run PostProcess= 0
Run WQNet= 0
UNET Theta= 0
UNET Theta Warmup= 0
UNET ZTol= 0
UNET ZSATol= 0
UNET MxIter= 0
UNET MaxInSteps= 0
UNET DtIC= 0
UNET DtMin= 0
UNET MaxCRTS= 0
UNET WFStab= 0
UNET SFStab= 0
UNET WFX= 1
UNET SFX= 1
UNET DSS MLevel= 1
UNET DZMax Abort= 0
UNET Convert EG Bridges= 0
UNET Use Existing IB Tables= 0
UNET Froude Reduction=False
UNET Froude Limit= 0
UNET Froude Power= 0
UNET Time Slicing=0,0, 5
DSS File=dss
Write IC File= 0
Echo Input=False
Echo Output=False
Write Detailed= 0
Detailed Automatic Start=False, 0
WQ ULTIMATE=-1
WQ Max Comp Step=1HOUR
WQ Output Interval=15MIN
WQ Output Selected Increments= 0
WQ Output face flow=0
WQ Output face velocity=0
WQ Output face area=0
WQ Output face dispersion=0
WQ Output cell volume=0
WQ Output cell surface area=0
WQ Output cell continuity=0
WQ Output face conc=0
WQ Output face dconc_dx=0
WQ Output face courant=0
WQ Output face peclet=0
WQ Output face adv mass=0
WQ Output face disp mass=0
WQ Output cell mass=0
WQ Output cell source sink temp=0
WQ Output cell source sink nsm=0
WQ Output MaxMinRange=-1
WQ Daily Max Min Mean=-1
WQ Daily Range=0
WQ Daily Time=0
WQ Create Restart=0
WQ Fixed Restart=0
WQ System Summary=False
Sorting and Armoring Iterations= 10
XS Update Threshold= 0.02
Hydraulics Update Threshold= 0.02
Energy Slope Method= 1
Volume Change Method= 0
XS Weighting Method= 0
Number of US Weighted Cross Sections= 1
Number of DS Weighted Cross Sections= 1
Upstream XS Weight=0.25
Main XS Weight=0.5
Downstream XS Weight=0.25
Number of DS XS's Weighted with US Boundary= 1
Upstream Boundary Weight= 1
Weight of XSs Associated with US Boundary= 0
Number of US XS's Weighted with DS Boundary= 1
Downstream Boundary Weight= 0.5
Weight of XSs Associated with DS Boundary= 0.5
Sediment Output Level= 4
Mass or Volume Output= 0
Output Increment Type= 1
Profile and TS Output Increment= 10
XS Output Flag= 0
XS Output Increment= 10
Disregard all LS=0
Disregard all Conn=0
Disregard all Breaches=0
Disregard all Pumps=0

--- smsfrk.f01 (steady flow) ---

Flow Title=USGS Regression Equation
Program Version=4.00
Number of Profiles= 1
Profile Names=P100yr
River Rch & RM=smsfrk,Main            ,19902.7
     430
River Rch & RM=smsfrk,Main            ,19103.5
     440
River Rch & RM=smsfrk,Main            ,18308.2
     486
River Rch & RM=smsfrk,Main            ,17517
     519
River Rch & RM=smsfrk,Main            ,15526.5
     563
River Rch & RM=smsfrk,Main            ,15240.2
     732
River Rch & RM=smsfrk,Main            ,13591.5
     800
River Rch & RM=smsfrk,Main            ,10714.6
     866
River Rch & RM=smsfrk,Main            ,10433.5
    1052
River Rch & RM=smsfrk,Main            ,9482.8
    1063
River Rch & RM=smsfrk,Main            ,6018.7
    1178
River Rch & RM=smsfrk,Main            ,255.7
    1308
Boundary for River Rch & Prof#=smsfrk,Main            , 1
Up Type= 0
Dn Type= 3
Dn Slope=0.018
DSS Import GetInterval= 0
DSS Import GetPeak= 0
DSS Import FillOption= 0

--- smsfrk.g01 (geometry) ---

Geom Title=USGS 3m DEM
Program Version=4.00

River Reach=smsfrk          ,Main
Reach XY= 30
     1712479.344      197175.535     1711462.417      196540.118
     1710925.754      195205.542     1710541.406      193486.712
     1709782.373      192779.212     1709102.717      192476.211
     1708098.972      192216.647     1707496.271      192299.233
      1706789.24      192730.223     1705934.599      192957.429
     1705863.459      193089.598     1705550.958      193016.681
     1705239.761      193188.556     1704806.167      193208.087
     1704569.187      193016.681     1703993.667      192094.806
     1704097.833      191433.348        1703877.      190877.659
     1703671.456       190698.58     1703433.771      190656.004
     1703298.354      190529.702     1703321.792      190415.119
     1702426.083      189914.854     1702130.386      189120.848
     1701396.503      188527.766     1701035.774      187792.352
     1700715.842      187619.502     1700036.636      187765.379
      1699684.87      187510.625     1699560.073      187692.462

Type RM Length L Ch R = 1 ,19902.7 ,407,398.5,390.1
XS GIS Cut Line= 4
     1712683.724      196994.268     1712371.638      197249.154
     1712360.462      197258.575     1712339.848      197554.862
#Sta/Elev= 30
    10.1 1248.09    20.1 1242.93    60.4 1229.13    90.7 1220.18   100.7 1220.17
   110.8 1214.66   120.9  1210.8     141 1204.97   161.2 1202.32   221.6 1201.42
   277.1 1194.68   282.1  1194.5   287.1 1194.85   302.2 1196.68   332.4 1198.12
   342.5 1201.47   362.7  1211.3   392.9 1232.15   402.9 1241.06   410.3  1245.1
   417.6 1247.64   486.9 1257.91   526.5 1260.66   536.4 1262.84   595.8 1291.09
   605.7 1292.55   635.4 1302.78     675 1313.72   694.8 1318.01   714.6 1320.62
#Mann= 3 , 0 , 0
       0      .1       0   277.1    .045       0   287.1      .1       0
Bank Sta=277.1,287.1
XS Rating Curve= 0 ,0
Exp/Cntr=0.3,0.1

Type RM Length L Ch R = 1 ,19504.2 ,399.7,400.7,401.6
XS GIS Cut Line= 3
     1712281.055      196684.579     1712158.967      196928.758
     1712036.878      197172.937
#Sta/Elev= 30
    10.1 1293.82    20.2 1289.72    30.3 1286.42    40.4 1284.01      91 1262.51
   141.6 1239.11   151.7 1238.07   171.9 1228.62     182 1222.98   202.2 1210.11
   222.4 1199.18   232.6 1194.88   262.9 1191.08     273 1187.93   278.1 1187.24
   283.1 1186.58   288.2 1186.83   333.7 1190.72   343.8 1196.41   353.9 1204.02
     364 1207.32   384.2 1217.32   394.3 1221.17   424.7 1231.04   465.1 1252.51
   485.3 1258.89   495.4 1265.22   515.7 1276.41   525.8 1280.84     546 1286.56
#Mann= 3 , 0 , 0
       0      .1       0   278.1    .045       0   288.2      .1       0
Bank Sta=278.1,288.2
XS Rating Curve= 0 ,0
Exp/Cntr=0.3,0.1

Type RM Length L Ch R = 1 ,19103.5 ,202.1,202.2,202.2
XS GIS Cut Line= 3
     1711934.361      196514.415      1711800.52      196752.356
     1711666.679      196990.296
#Sta/Elev= 30
    10.1  1300.7    70.8 1266.23    80.9 1264.04      91 1258.86   101.1 1251.07
   111.2 1241.89   121.3  1230.5   131.4 1217.33   141.6  1205.7   151.7 1198.15
   161.8  1192.7   171.9 1189.13     182 1187.15   202.2 1185.41   212.3 1185.35
   242.7 1186.97   252.8 1186.05   267.9 1181.19     273 1179.76   278.1 1179.97
   303.3 1181.74   313.4 1184.22   323.6 1188.22   384.2 1217.01   404.4  1228.1
   424.7 1233.27   505.6 1272.39   515.7 1276.93   525.8  1277.7     546 1288.54
#Mann= 3 , 0 , 0
       0      .1       0   267.9    .045       0   278.1      .1       0
Bank Sta=267.9,278.1
XS Rating Curve= 0 ,0
Exp/Cntr=0.3,0.1

Type RM Length L Ch R = 1 ,18901.4 ,305.3,320.9,336.4
XS GIS Cut Line= 3
     1711823.153      196406.342     1711708.095      196507.031
     1711482.879      196904.023
#Sta/Elev= 30
     9.6 1319.55    47.8 1293.01    66.9 1275.66    76.4 1270.27    95.6 1262.93
   114.7 1253.19   133.8  1245.7   143.3 1240.79   162.8 1219.24   182.7 1200.14
   192.6 1191.79   202.5 1186.42   212.4 1184.04   222.4 1183.39   242.2 1179.76
   291.8 1179.59   316.4 1173.86   321.6 1173.41   326.7 1173.48   351.3  1175.4
   361.3 1178.21     391  1191.9     401 1194.35   420.8 1194.43   440.6 1196.87
   450.6  1200.4   500.2 1225.63   549.8 1252.75   559.7 1254.51   609.3 1284.94
#Mann= 3 , 0 , 0
       0      .1       0   316.4    .045       0   326.7      .1       0
Bank Sta=316.4,326.7
XS Rating Curve= 0 ,0
Exp/Cntr=0.3,0.1

Type RM Length L Ch R = 1 ,18580.5 ,273.6,272.3,270.9
XS GIS Cut Line= 4
      1711673.74      196339.072     1711534.411      196394.422
     1711236.667      196482.219     1711078.252       196783.78
#Sta/Elev= 30
      10 1269.75      50 1260.07      70 1251.88    99.9 1243.48   109.9 1239.18
   129.9 1228.44   139.9 1219.02   149.9 1212.92     180  1197.3     200 1188.05
     220 1176.95     230 1173.88   250.1 1171.54   274.9 1166.81   280.1 1166.14
   285.3 1166.27   290.1 1166.38   300.1  1169.2   310.1 1170.49   360.2  1173.9
   420.3 1179.81   440.3 1183.45   490.4 1195.29   510.4 1198.04   540.5 1204.42
   600.6 1219.38   730.8 1224.09   750.9 1226.18   770.9 1231.79     801 1243.64
#Mann= 3 , 0 , 0
       0      .1       0   274.9    .045       0   285.3      .1       0
Bank Sta=274.9,285.3
XS Rating Curve= 0 ,0
Exp/Cntr=0.3,0.1

Type RM Length L Ch R = 1 ,18308.2 ,246.4,245.5,244.5
XS GIS Cut Line= 3
     1711531.601       196096.77     1711275.288      196190.751
     1711018.975      196284.733
#Sta/Elev= 30
    10.1 1282.49    40.4 1265.15    70.8 1248.65    80.9 1243.68      91 1236.51
   101.1 1229.65   141.6 1210.81   151.7 1205.73   161.8 1199.96   171.9 1187.81
   192.1 1171.59   202.2 1166.38   222.4 1162.08   232.6 1159.62   237.5  1159.5
   242.7 1159.37   247.9 1160.36     273 1165.31   303.3 1170.48   323.6 1173.41
   333.7 1175.27   353.9 1176.91   394.3 1179.14   404.4 1181.94   414.6 1185.93
   465.1 1207.31   475.2 1212.41   485.3 1221.29   515.7 1235.17     546  1248.6
#Mann= 3 , 0 , 0
       0      .1       0   237.5    .045       0   247.9      .1       0
Bank Sta=237.5,247.9
XS Rating Curve= 0 ,0
Exp/Cntr=0.3,0.1

Type RM Length L Ch R = 1 ,18062.7 ,264.6,266.3,268
XS GIS Cut Line= 3
      1711442.59      195855.836     1711191.308      195962.545
     1710940.027      196069.253
#Sta/Elev= 30
    10.1 1212.59    20.2 1208.53    30.3 1205.89    50.6 1202.53    70.8 1194.97
    80.9 1190.24      91 1183.95   101.1 1172.57   111.2 1168.79   121.3  1166.7
   161.8  1162.3     182 1159.19   222.4 1156.04   237.4 1153.12   242.7 1152.43
   247.9 1152.73   252.8 1153.02   262.9 1155.39   293.2 1160.14   303.3 1162.65
   333.7 1172.27   343.8 1177.66   374.1 1186.07   384.2  1189.8   404.4 1198.72
   424.7 1212.33   475.2 1234.44   495.4 1242.37   505.6 1248.65     546 1263.36
#Mann= 3 , 0 , 0
       0      .1       0   237.4    .045       0   247.9      .1       0
Bank Sta=237.4,247.9
XS Rating Curve= 0 ,0
Exp/Cntr=0.3,0.1

Type RM Length L Ch R = 1 ,17796.4 ,280.1,279.4,278.7
XS GIS Cut Line= 2
      1711328.26      195635.736     1710867.647      195785.881
#Sta/Elev= 30
    10.1  1175.7    30.3 1170.87    40.4 1169.43    60.6 1168.51    70.7  1167.7
    90.8 1164.61   141.3 1158.72   161.5 1154.84   171.6 1153.76   191.8 1152.82
   201.9 1151.12     212 1148.51   216.8 1147.92     222 1147.27   227.3 1148.11
   252.3 1152.35   262.4 1154.59   272.5  1157.8   302.8 1168.64     323 1179.25
   353.3 1190.29   363.3  1194.8   373.4 1200.93   383.5 1208.88   393.6  1221.4
   423.9 1240.88   454.2 1256.93   464.3  1265.9   474.4 1273.06   484.5 1278.88
#Mann= 3 , 0 , 0
       0      .1       0   216.8    .045       0   227.3      .1       0
Bank Sta=216.8,227.3
XS Rating Curve= 0 ,0
Exp/Cntr=0.3,0.1

Type RM Length L Ch R = 1 ,17517   ,296.4,301.1,305.8
XS GIS Cut Line= 3
     1711238.752      195362.505     1710982.575      195456.612
     1710721.152      195536.929
#Sta/Elev= 30
    10.1 1218.12    30.3 1205.61    40.4 1201.58    50.5 1198.23    60.6 1193.43
    70.8  1188.2      91 1174.95   101.1 1171.14   141.5  1158.1   161.7 1152.66
   171.8 1151.26   181.9 1150.82   192.1 1149.73   222.4 1144.37   227.2 1143.93
   232.5 1143.44   237.8 1143.84   272.9 1148.56     283 1150.76   303.3 1158.18
   313.4 1161.37   323.6 1169.88   353.9 1185.76   394.5 1206.03   404.6 1213.54
   414.7 1219.69   465.4 1244.65   475.5 1251.52   485.6 1259.68   546.4 1292.12
#Mann= 3 , 0 , 0
       0      .1       0   227.2    .045       0   237.8      .1       0
Bank Sta=227.2,237.8
XS Rating Curve= 0 ,0
Exp/Cntr=0.3,0.1

Type RM Length L Ch R = 1 ,17215.9 ,268.3,268.8,269.3
XS GIS Cut Line= 3
     1711144.392      195133.711     1710873.318      195166.078
     1710602.243      195198.446
#Sta/Elev= 30
    10.1 1238.42    70.8 1205.21    80.9 1197.57      91 1186.19   111.2 1175.83
   151.7 1157.89   161.8 1149.87   171.9 1146.74   192.1 1142.97   202.2 1138.42
   212.3 1134.84   217.1 1134.67   222.4 1134.48   227.8 1135.06   242.7 1138.06
   262.9  1140.4   283.1 1144.83   303.3 1151.88   313.4 1161.02   333.7 1171.14
   343.8 1174.36   374.1 1177.27   384.2 1178.89   394.3 1183.63   424.7 1191.93
     455 1201.45   465.1 1206.78   505.6 1219.61   535.9 1230.15     546 1235.79
#Mann= 3 , 0 , 0
       0      .1       0   217.1    .045       0   227.8      .1       0
Bank Sta=217.1,227.8
XS Rating Curve= 0 ,0
Exp/Cntr=0.3,0.1

Type RM Length L Ch R = 1 ,16947.1 ,207.5,208.9,210.2
XS GIS Cut Line= 2
     1711068.688      194877.379     1710681.875      194913.006
#Sta/Elev= 30
      10 1223.77    19.9 1218.54    29.9  1209.7    39.8 1202.84    89.6 1176.77
    99.6 1168.69   109.6 1161.04   129.5 1150.54   139.4 1145.36   149.4 1141.15
   159.4 1138.56   169.3 1136.37   179.3 1133.16   183.9 1132.41   189.2 1131.54
   194.6 1132.65   209.2 1135.58   229.1 1139.25     239 1141.54     249 1144.15
     259 1147.13   268.9 1148.48   278.9 1150.14   288.8 1152.37   298.8 1155.02
   308.8 1158.08   318.7 1161.49   328.7 1165.33   338.6 1172.61   388.5 1189.36
#Mann= 3 , 0 , 0
       0      .1       0   183.9    .045       0   194.6      .1       0
Bank Sta=183.9,194.6
XS Rating Curve= 0 ,0
Exp/Cntr=0.3,0.1

Type RM Length L Ch R = 1 ,16738.2 ,243.4,241.4,239.4
XS GIS Cut Line= 3
     1711093.043       194681.93     1710790.289      194689.982
     1710551.104      194663.545
#Sta/Elev= 30
    10.1 1240.19    40.4  1223.9    60.6 1211.87    80.8 1193.52     101 1182.66
     111 1178.23   131.2 1170.97   141.3 1165.52   151.4 1157.28   191.8 1137.55
   201.9    1134   222.1 1131.03   232.2 1127.03   236.9 1126.35   242.3 1125.58
   247.7 1125.82   252.4 1126.03   272.6 1130.93   292.8 1134.11   312.9 1143.05
     343 1157.77     353 1160.94     373 1164.23   383.1 1166.91   443.2 1175.47
   453.3  1179.6   503.4    1191   523.4 1196.47   533.5 1202.96   543.5 1207.68
#Mann= 3 , 0 , 0
       0      .1       0   236.9    .045       0   247.7      .1       0
Bank Sta=236.9,247.7
XS Rating Curve= 0 ,0
Exp/Cntr=0.3,0.1

Type RM Length L Ch R = 1 ,16496.8 ,167.7,167,166.3
XS GIS Cut Line= 2
     1710984.709       194429.49     1710580.082      194480.386
#Sta/Elev= 30
     9.9 1157.47    29.8 1151.12    39.8 1147.42    49.7  1142.3    59.7 1133.64
    69.6 1130.98    79.6 1129.65    89.5 1128.99    99.5 1128.78   139.3 1128.74
   149.2 1128.27   159.1 1126.78   169.1  1124.3     179 1122.24   183.6 1122.05
     189 1121.83   194.4 1122.55   198.9 1123.16   208.9 1125.87   218.8 1128.11
   228.8 1130.17   238.7 1134.18   278.5 1154.02   288.5 1159.33   298.4 1163.01
   338.2 1174.62   348.1 1177.69   358.1 1181.24     368 1187.62   407.8 1200.49
#Mann= 3 , 0 , 0
       0      .1       0   183.6    .045       0   194.4      .1       0
Bank Sta=183.6,194.4
XS Rating Curve= 0 ,0
Exp/Cntr=0.3,0.1

Type RM Length L Ch R = 1 ,16329.8 ,402.2,400,397.8
XS GIS Cut Line= 3
     1711035.881      194245.604      1710766.31      194288.735
     1710496.739      194331.866
#Sta/Elev= 30
    10.1 1153.98    40.4 1148.08    50.6 1144.88    60.7  1143.6    70.8 1142.97
   111.2 1142.44   121.3 1140.87   141.6 1136.73   171.9 1129.14     182 1127.72
   202.2 1126.15   257.4 1119.79   262.9 1119.25   268.3 1119.98     273 1120.62
   283.1  1123.3   303.3 1126.77   313.4 1130.96   343.8 1148.75     364 1163.02
   374.1 1165.98   414.6 1174.44   424.7  1177.8   434.8 1182.28   444.9 1185.81
   475.2 1200.82   485.3 1204.06   505.6 1209.18   515.7  1212.3     546 1218.27
#Mann= 3 , 0 , 0
       0      .1       0   257.4    .045       0   268.3      .1       0
Bank Sta=257.4,268.3
XS Rating Curve= 0 ,0
Exp/Cntr=0.3,0.1

Type RM Length L Ch R = 1 ,15929.8 ,406.7,403.4,400.1
XS GIS Cut Line= 3
     1710929.758      193828.873     1710666.637      193901.651
     1710403.517      193974.429
#Sta/Elev= 30
    10.1 1222.36    40.4  1205.2    50.6 1198.23    60.7 1188.85      91  1173.4
   121.3 1159.36   131.4 1149.96   171.9 1129.66     182  1125.4   192.1 1123.14
   212.3 1122.13   242.7 1118.83   262.9 1113.84   267.5 1113.13     273 1112.29
   278.5 1112.75   283.1 1113.14   293.2 1114.89   303.3 1114.97   313.4 1115.84
   353.9 1124.07     364  1127.6   384.2 1132.14   394.3 1135.83   434.8 1153.84
   444.9  1160.4     455 1164.94   505.6 1183.29   525.8 1193.71     546 1201.72
#Mann= 3 , 0 , 0
       0      .1       0   267.5    .045       0   278.5      .1       0
Bank Sta=267.5,278.5
XS Rating Curve= 0 ,0
Exp/Cntr=0.3,0.1

Type RM Length L Ch R = 1 ,15526.5 ,294.8,286.3,277.9
XS GIS Cut Line= 3
     1710781.055      193409.681     1710533.489      193524.747
     1710285.923      193639.813
#Sta/Elev= 30
    10.1 1146.33    20.2 1139.21    50.6 1127.26    70.8 1121.02      91 1116.32
   101.1 1113.52   121.3 1111.98   131.4 1111.79   171.9 1112.52   192.1 1111.99
   247.2 1105.55   252.8 1104.98   258.3 1105.72   262.9 1106.35     273 1109.54
   283.1 1112.12   293.2 1113.27   333.7 1115.52   343.8 1116.76   353.9 1118.87
   374.1 1125.71   384.2  1129.5   404.4 1138.36   414.6 1143.85   424.7  1151.8
   495.4 1184.89   505.6 1190.77   515.7 1197.78   525.8 1202.37     546 1212.43
#Mann= 3 , 0 , 0
       0     .08       0   247.2    .045       0   258.3      .1       0
Bank Sta=247.2,258.3
XS Rating Curve= 0 ,0
Exp/Cntr=0.3,0.1

Type RM Length L Ch R = 1 ,15240.2 ,196.4,191.7,186.9
XS GIS Cut Line= 3
     1710595.351      193045.106     1710310.331      193373.388
     1710228.038      193519.869
#Sta/Elev= 30
    10.1 1186.85    30.3 1174.43    40.4 1169.49    60.7 1162.58   101.1 1151.45
   111.2 1147.14   131.4 1136.36   141.5 1132.04   151.7 1131.07   161.8 1127.18
   192.1 1112.49   202.2 1109.03   242.7 1103.53   283.1 1101.83   328.1 1097.67
   333.6 1097.63   339.2 1098.97     364 1105.24   384.2 1109.08   394.3 1109.63
   404.4 1111.39   424.6 1115.92   434.7 1119.93   454.5 1131.94   503.9 1156.39
   513.8 1158.23   523.7 1161.71   563.2 1181.51     583 1192.52   602.8 1201.39
#Mann= 3 , 0 , 0
       0      .1       0   328.1    .045       0   339.2      .1       0
Bank Sta=328.1,339.2
XS Rating Curve= 0 ,0
Exp/Cntr=0.3,0.1

Type RM Length L Ch R = 1 ,15048.5 ,209.9,217.5,225
XS GIS Cut Line= 3
     1710351.048      193012.023     1710282.338      193065.464
     1710127.104      193365.754
#Sta/Elev= 30
     9.7 1155.09      29 1147.09    38.7 1145.68    48.4 1143.49      58 1139.26
    77.4 1129.26      87 1122.94      97 1115.86   106.9 1109.52   116.9 1103.74
   126.8 1098.89   136.8  1097.3   186.5 1097.15   196.4 1096.24   210.7 1093.04
   216.3 1091.76   221.9 1091.82   226.2 1091.87   236.2 1093.84   246.1 1096.71
     266 1101.07     276 1101.73   325.7 1116.45   335.6  1119.9   345.5 1124.03
   365.4 1132.71   375.4 1137.78   385.3 1140.32   395.3 1143.55   425.1 1156.66
#Mann= 3 , 0 , 0
       0      .1       0   210.7    .045       0   221.9      .1       0
Bank Sta=210.7,221.9
XS Rating Curve= 0 ,0
Exp/Cntr=0.3,0.1

Type RM Length L Ch R = 1 ,14831   ,166.7,161.8,156.9
XS GIS Cut Line= 4
     1710312.896      192898.908     1710129.668      192990.522
      1709955.03      193143.688     1709936.421      193229.576
#Sta/Elev= 30
     9.8 1187.53    19.5 1182.56    48.8 1169.36    68.3 1165.04    87.8 1158.55
   117.1 1150.18   146.3 1140.74   185.3 1125.99   225.1 1108.02   235.2 1105.24
   245.3 1104.42   255.4 1102.67   285.7 1096.34   295.8 1093.98   305.9  1090.3
   310.3 1089.63   315.9 1088.78   321.6 1090.38   336.1 1094.04   356.3 1094.98
   386.6 1094.61   406.8 1096.81   416.9 1098.89   437.1 1104.19   456.7 1111.37
   466.4 1115.53   495.7 1131.05   505.5 1132.17   515.3 1136.03     525 1140.63
#Mann= 3 , 0 , 0
       0      .1       0   310.3    .045       0   321.6      .1       0
Bank Sta=310.3,321.6
XS Rating Curve= 0 ,0
Exp/Cntr=0.3,0.1

Type RM Length L Ch R = 1 ,14669.2 ,158.7,166.5,174.3
XS GIS Cut Line= 3
     1710135.763      192805.784     1709962.187      192904.634
     1709757.326      193199.358
#Sta/Elev= 30
      10 1207.32      20 1203.71      30 1197.63    39.9  1190.4    99.9 1162.04
   109.9 1156.82   119.8 1150.19   149.8 1137.29   179.8 1125.61   189.8 1122.69
   199.7 1121.78   209.7 1115.53   229.7 1105.69   239.6 1099.66   249.6 1091.25
   259.6 1085.16   263.9 1084.49   269.5 1083.61   275.2 1084.66   279.5 1085.45
   289.5 1089.18   299.5 1091.16   359.3 1092.63   379.2 1094.53     439 1105.71
   498.9 1149.57   528.8 1169.88   538.7  1175.7   548.7 1177.56   558.7 1183.81
#Mann= 3 , 0 , 0
       0      .1       0   263.9    .045       0   275.2      .1       0
Bank Sta=263.9,275.2
XS Rating Curve= 0 ,0
Exp/Cntr=0.3,0.1

Type RM Length L Ch R = 1 ,14502.7 ,413.4,402.6,391.8
XS GIS Cut Line= 3
     1710015.131      192709.189     1709691.939      192920.409
     1709451.631      192966.886
#Sta/Elev= 30
     9.9 1200.12    79.2 1149.72    89.1 1140.64      99 1135.19   138.6 1115.78
   158.4 1109.77   178.2 1098.84   207.9 1086.35   217.8 1082.41   227.7 1080.36
   231.9 1080.22   237.6 1080.03   243.3 1080.99   247.5  1081.7   257.4 1085.82
   267.3 1087.05     297 1088.64   326.7 1088.73   395.9 1090.99   415.5 1093.54
     435 1100.98   493.8 1118.57   503.6  1122.1   523.2 1127.28   532.9 1130.84
   572.1    1147   581.9 1153.11   591.7 1157.78   601.5 1160.78   630.9 1172.77
#Mann= 3 , 0 , 0
       0      .1       0   231.9    .045       0   243.3      .1       0
Bank Sta=231.9,243.3
XS Rating Curve= 0 ,0
Exp/Cntr=0.3,0.1

Type RM Length L Ch R = 1 ,14100.2 ,219.9,220.5,220.6
XS GIS Cut Line= 2
     1709574.877      192480.155     1709399.284      192816.072
#Sta/Elev= 30
      10 1134.03    29.9 1121.79    39.9 1115.91    59.8 1102.34    69.8 1096.56
    79.8  1094.6    89.8 1090.37    99.7 1085.52   109.7  1082.7   119.7  1081.8
   169.6  1078.7   179.5 1077.46   189.5 1075.94   203.7  1074.4   209.5 1073.86
   215.2 1075.79   219.4 1077.21   229.4 1081.06   239.4 1082.35   269.3 1082.51
   279.3 1083.38   289.3 1086.69   299.2  1091.2   309.2 1092.28   319.2 1095.77
   329.2 1100.27   339.1 1105.64   349.1 1112.36   369.1 1123.46     379  1129.4
#Mann= 3 , 0 , 0
       0      .1       0   203.7    .045       0   215.2      .1       0
Bank Sta=203.7,215.2
XS Rating Curve= 0 ,0
Exp/Cntr=0.3,0.1

Type RM Length L Ch R = 1 ,13879.7 ,293.8,288.2,282.9
XS GIS Cut Line= 3
     1709437.901      192308.271     1709295.227      192540.891
     1709166.829       192782.53
#Sta/Elev= 30
    10.1 1164.53    20.2 1158.03    30.3 1153.46    40.4 1150.52    60.6  1138.3
   101.1 1115.65   121.3 1101.68   131.4 1095.83   141.5 1093.46   151.6 1089.54
   161.7 1084.48   171.8 1081.39   181.9 1080.43   222.4 1079.16   262.8 1075.52
   272.9 1071.45   277.3 1070.25     283 1068.69   288.8 1069.15   293.2  1069.5
   313.4 1076.82   323.6 1077.46   374.2 1078.09   384.4 1079.75   394.5 1084.86
   475.6 1137.62   485.7 1142.38   495.8 1144.58   516.1 1159.27   546.5  1177.7
#Mann= 3 , 0 , 0
       0      .1       0   277.3    .045       0   288.8      .1       0
Bank Sta=277.3,288.8
XS Rating Curve= 0 ,0
Exp/Cntr=0.3,0.1

Type RM Length L Ch R = 1 ,13591.5 ,167.7,167.4,167.2
XS GIS Cut Line= 4
     1709141.422      192098.392     1709046.945      192338.877
     1708988.255      192593.678     1709028.336      192723.941
#Sta/Elev= 30
     9.9  1126.8    29.8 1127.13    39.8 1130.95    49.7 1130.25    59.6 1127.66
    79.5 1119.56   109.3  1102.5   119.3 1102.73   139.1 1091.99   149.1 1088.37
   168.9 1082.93   188.8 1078.88   218.6 1075.22   288.5  1070.7   358.9  1071.3
     369 1069.71   383.3 1063.99   389.1 1062.18   394.9 1063.81   399.2 1065.02
   409.2 1070.18   419.3    1073   459.5 1072.77   469.6 1074.95   529.6  1109.6
   539.3 1110.03   549.1 1114.04   636.7 1161.32   646.4    1161   656.1 1165.04
#Mann= 3 , 0 , 0
       0      .1       0   383.3    .045       0   394.9      .1       0
Bank Sta=383.3,394.9
XS Rating Curve= 0 ,0
Exp/Cntr=0.3,0.1

Type RM Length L Ch R = 1 ,13424.1 ,394.7,397.5,400.3
XS GIS Cut Line= 3
     1708925.271      192112.706     1708835.089      192523.536
      1708834.97      192696.633
#Sta/Elev= 30
      10 1170.37    40.1 1148.04    60.1 1134.89    70.1 1130.44    80.1 1128.92
   110.2 1108.82   140.2 1094.09   170.2 1081.32   180.3 1080.96   210.3 1071.83
   240.3 1065.96   260.4  1064.7   290.4  1065.9   300.4 1064.84   314.7 1061.78
   320.5 1060.89   326.3 1061.77   330.5 1062.42   340.5 1066.36   350.5 1068.92
   390.6 1070.98   400.6 1072.81   410.6 1076.77   478.3 1113.53   487.9 1115.02
   497.5 1118.57     536  1140.5   574.5 1163.84   584.1 1168.73   593.7 1169.37
#Mann= 3 , 0 , 0
       0     .08       0   314.7    .045       0   326.3      .1       0
Bank Sta=314.7,326.3
XS Rating Curve= 0 ,0
Exp/Cntr=0.3,0.1

Type RM Length L Ch R = 1 ,13026.6 ,384.4,375.6,366.7
XS GIS Cut Line= 3
     1708567.405       192076.92      1708425.69      192456.258
     1708473.953       192627.12
#Sta/Elev= 30
    10.1 1161.59    70.9 1121.91    91.1 1116.16   131.6 1089.43   141.7 1083.69
     162 1073.25   172.1 1070.04   182.2 1067.92     243  1061.9   253.1 1060.26
   273.3 1054.94   277.6 1054.54   283.5 1053.99   289.3 1055.26   293.6  1056.2
   303.7 1056.74   313.8 1061.51     324 1063.14   384.7 1063.74   404.9 1068.15
   414.8 1073.33   424.7  1083.1   434.5 1093.81   444.4 1103.55   454.3 1111.18
   464.1 1116.68   503.6 1135.18   513.4 1136.14   523.3 1139.25   582.5 1167.76
#Mann= 3 , 0 , 0
       0      .1       0   277.6    .045       0   289.3      .1       0
Bank Sta=277.6,289.3
XS Rating Curve= 0 ,0
Exp/Cntr=0.3,0.1

Type RM Length L Ch R = 1 ,12651   ,384.6,381.1,377.6
XS GIS Cut Line= 3
     1708102.179        191989.6     1708130.809      192397.568
     1708100.008      192565.652
#Sta/Elev= 30
      10 1117.11    19.9 1113.29    29.9 1111.65    49.9 1101.64    69.8 1092.42
    89.8 1083.85   109.7 1076.43   119.7 1073.48   129.7 1073.09   179.5 1058.23
   219.4 1048.26   233.5 1047.95   239.4 1047.66   245.3 1050.02   259.3 1056.26
   269.3 1057.51   339.1 1058.02   349.1  1058.9   359.1  1061.9     399 1080.62
   429.1 1095.26   449.2  1100.1   469.3 1109.77   489.4 1120.86   509.5 1132.92
   529.6 1145.54   539.6 1150.17   549.7 1151.98   559.7 1158.01   579.9 1169.33
#Mann= 3 , 0 , 0
       0      .1       0   233.5    .045       0   245.3      .1       0
Bank Sta=233.5,245.3
XS Rating Curve= 0 ,0
Exp/Cntr=0.3,0.1

Type RM Length L Ch R = 1 ,12269.9 ,420.6,413.4,406.3
XS GIS Cut Line= 3
     1707725.631      191998.675     1707724.273      192192.868
     1707804.435      192523.536
#Sta/Elev= 30
     9.7 1126.39    48.5 1103.14    77.7 1086.76    87.4 1086.29   116.5 1073.22
   135.9  1065.6   155.4 1058.87   165.1 1056.57   174.8  1055.2   194.2 1054.24
   244.2 1048.92   264.2 1044.21   268.3 1043.86   274.3 1043.34   280.2  1044.3
   284.3 1044.97   294.3 1045.07   304.3 1047.66   324.3 1048.73   334.3 1050.05
   354.3 1055.72   364.3  1060.7   394.3 1077.86   414.4 1085.69   424.4 1092.33
   444.4 1103.98   484.4 1123.69   504.4 1132.29   514.4 1133.18   534.4  1142.4
#Mann= 3 , 0 , 0
       0      .1       0   268.3    .045       0   280.2      .1       0
Bank Sta=268.3,280.2
XS Rating Curve= 0 ,0
Exp/Cntr=0.3,0.1

Type RM Length L Ch R = 1 ,11856.5 ,393,396.5,400
XS GIS Cut Line= 3
     1707205.789      192162.491     1707358.225      192388.968
     1707510.662      192615.446
#Sta/Elev= 30
    10.1  1172.5    20.2 1164.61    30.3 1155.16    40.4 1147.36      91 1113.81
   101.1 1110.68   111.2 1105.57   121.3 1099.41   131.4 1094.41   151.7 1085.64
   171.9 1075.73     182 1071.56   202.2 1060.74   222.4 1051.76   242.7 1046.46
   252.8 1041.16   256.9 1039.91   262.9 1038.07   268.9 1038.22     273 1038.31
   293.2 1042.13   303.3 1043.24   394.3 1046.49   404.4 1048.57   414.6  1052.9
   485.3 1091.49   495.4 1097.62   505.6 1100.07   515.7 1103.76     546 1117.26
#Mann= 3 , 0 , 0
       0      .1       0   256.9    .045       0   268.9      .1       0
Bank Sta=256.9,268.9
XS Rating Curve= 0 ,0
Exp/Cntr=0.3,0.1

Type RM Length L Ch R = 1 ,11460   ,397.9,399.3,400.8
XS GIS Cut Line= 3
     1706904.789      192335.817     1707015.334      192585.434
     1707125.879      192835.051
#Sta/Elev= 30
    10.1  1171.6    30.3 1158.88    50.6 1148.22    60.7 1142.37      91 1123.48
   101.1 1121.42   111.2 1117.42   141.6 1097.32   171.9 1076.44   202.2 1057.38
   212.3  1055.5   222.4 1051.62   252.8 1034.07   256.8 1033.04   262.9 1031.47
     269 1032.23     273 1032.73   283.1 1035.94   293.2 1037.54   313.4 1039.26
   394.3 1039.31   414.6 1041.98   424.7 1045.04   434.8 1048.96   444.9 1050.75
     455 1053.43   485.3 1065.17   505.6 1074.23   515.7  1079.2     546 1095.97
#Mann= 3 , 0 , 0
       0      .1       0   256.8    .045       0     269      .1       0
Bank Sta=256.8,269
XS Rating Curve= 0 ,0
Exp/Cntr=0.3,0.1

Type RM Length L Ch R = 1 ,11060.7 ,344,346.1,348.2
XS GIS Cut Line= 3
     1706578.486      192526.714     1706671.973       192783.23
     1706762.616      193040.739
#Sta/Elev= 30
    10.1 1174.87    30.3  1164.1    40.4 1157.52    50.6 1150.11    60.7 1141.59
    70.8 1132.19    80.9 1130.29      91 1121.58   111.2 1101.01   121.3 1091.66
   131.5 1083.42   141.6 1076.13   151.7 1069.65   171.9  1058.4     182 1053.97
   192.1 1050.18   202.2 1047.95   232.6 1032.52   242.7 1028.92   246.7 1028.61
   252.8 1028.15   258.9 1029.43     273    1033   293.2 1035.73   424.7 1037.24
   495.5 1042.19   505.6 1044.04   525.8 1052.31   535.9 1055.01     546 1058.63
#Mann= 3 , 0 , 0
       0      .1       0   246.7    .045       0   258.9      .1       0
Bank Sta=246.7,258.9
XS Rating Curve= 0 ,0
Exp/Cntr=0.3,0.1

Type RM Length L Ch R = 1 ,10714.6 ,283.3,281.1,278.9
XS GIS Cut Line= 3
     1706272.769      192606.561     1706358.657      192954.407
     1706421.641      193206.344
#Sta/Elev= 30
      10 1118.24    19.9 1114.81    39.8  1109.6    59.7  1101.1    69.7 1101.26
   119.4 1081.35   149.3 1070.66   169.2 1062.53   179.1 1059.94   189.1 1058.51
   199.1 1054.95     219 1049.64   238.9  1046.1   248.8 1038.84   258.8 1028.06
   262.6 1026.56   268.7 1024.16   274.9 1025.41   288.6 1026.52   298.6 1029.58
   308.5 1031.25   328.4 1032.67   468.2 1036.33   498.1 1033.78   528.1 1033.54
   538.1  1034.7   558.1 1041.18     578 1049.48     598 1059.12     618 1066.37
#Mann= 3 , 0 , 0
       0      .1       0   262.6    .045       0   274.9      .1       0
Bank Sta=262.6,274.9
XS Rating Curve= 0 ,0
Exp/Cntr=0.3,0.1

Type RM Length L Ch R = 1 ,10433.5 ,211.8,189.1,166.4
XS GIS Cut Line= 3
     1705976.456      192669.546      1706078.09      192950.112
     1706305.693      193119.025
#Sta/Elev= 30
     9.9 1138.59    49.7 1117.56    79.6 1100.45    89.5 1098.99    99.5 1094.78
   169.1 1055.29   198.9 1039.52   208.9 1038.58   218.8 1034.24   228.8 1028.15
   238.7 1022.63   242.5 1021.91   248.7 1020.74   254.9 1022.42   258.6 1023.42
   268.6 1027.86   278.5 1029.64   298.4 1029.74     349 1030.54   389.5 1031.71
     430 1032.39   460.4 1032.42   470.5 1033.29     511  1042.3   521.1  1043.6
   531.2 1043.38   541.4 1044.44   551.5 1046.01   561.6 1047.24   581.8 1048.06
#Mann= 3 , 0 , 0
       0      .1       0   242.5    .045       0   254.9      .1       0
Bank Sta=242.5,254.9
XS Rating Curve= 0 ,0
Exp/Cntr=0.3,0.1

Type RM Length L Ch R = 1 ,10244.4 ,65.3,66.1,67
XS GIS Cut Line= 4
     1705797.523      192809.829     1705800.386      192980.173
     1705969.299      193000.214     1706095.268      193216.365
#Sta/Elev= 30
      10 1089.36      20 1085.36    30.1 1084.05    60.1 1068.95    80.2 1059.54
   110.2  1047.6   130.3 1041.06   140.3 1040.64   150.3 1037.43   170.4 1032.52
   190.4 1031.65   200.4 1030.63   230.4 1026.05   260.4 1020.12   264.2  1019.7
   270.4 1019.01   276.6 1020.37   280.4 1021.21   290.4 1026.96   300.4 1027.86
   370.5 1028.34   420.5 1030.03   490.6 1035.74   500.6 1037.49   510.6 1040.54
   520.6 1044.19   530.6 1046.82   540.6 1047.73   570.6 1060.96   590.6 1070.42
#Mann= 3 , 0 , 0
      10      .1       0   264.2    .045       0   276.6      .1       0
#XS Ineff= 2 , 0
       0     230             285       0
Permanent Ineff=
       F       F
Bank Sta=264.2,276.6
XS Rating Curve= 0 ,0
Exp/Cntr=0.3,0.1

Type RM Length L Ch R = 1 ,10178.3 ,358.9,385,411.1
XS GIS Cut Line= 4
     1705711.636      192814.123     1705778.915      193038.863
     1705956.416      193067.492     1706017.969      193263.603
#Sta/Elev= 30
     9.8 1097.18    29.3 1092.25    78.2 1066.74    97.7 1057.02   117.3  1048.3
   127.1 1047.21   136.8 1044.52   156.4 1037.32   175.9 1031.31   185.7 1029.17
   205.3  1027.8   234.6 1027.17   304.5 1028.34   314.5 1026.43   334.5 1019.82
   338.2 1019.35   344.5 1018.56   350.7 1019.69   354.5 1020.39   374.4 1028.95
   414.4 1029.14   443.8 1031.13   492.7  1037.3   502.5 1039.89   512.3 1043.96
   522.1 1044.39   531.8 1047.95   541.6 1052.47   580.8 1071.96   619.9 1086.67
#Mann= 3 , 0 , 0
     9.8      .1       0   338.2    .045       0   350.7      .1       0
#XS Ineff= 2 , 0
       0     327             357       0
Permanent Ineff=
       F       F
Bank Sta=338.2,350.7
XS Rating Curve= 0 ,0
Exp/Cntr=0.3,0.1

Type RM Length L Ch R = 1 ,9793.2  ,313.6,310.4,307.2
XS GIS Cut Line= 3
     1705609.692      192748.452     1705535.566      192937.229
     1705594.289      193315.577
#Sta/Elev= 30
     9.7 1133.23    57.9 1116.42    67.6 1112.18    77.3 1109.75    86.9 1108.12
   164.2 1065.02   173.8 1061.23   183.5 1060.99   202.8 1051.71     223 1040.86
     233 1036.51   243.1 1034.06   253.2 1032.56   263.3  1027.2   273.3 1020.75
   283.4 1018.91   287.2  1018.9   293.5 1018.55   299.8 1019.87   313.6 1022.55
   323.7  1023.4   414.4 1024.46   424.5  1024.8   434.6 1026.34   444.6 1030.09
   484.9 1051.35     495 1054.96   505.1 1056.83   555.5 1085.33   585.7 1100.61
#Mann= 3 , 0 , 0
     9.7      .1       0   287.2    .045       0   299.8      .1       0
Bank Sta=287.2,299.8
XS Rating Curve= 0 ,0
Exp/Cntr=0.3,0.1

Type RM Length L Ch R = 1 ,9482.8  ,275.4,281,286.5
XS GIS Cut Line= 3
     1705190.574      192898.264     1705297.943      193230.679
     1705382.578      193417.369
#Sta/Elev= 30
      10 1105.91    29.9 1096.25    39.9 1093.28    49.9 1089.11    59.9 1082.89
    69.9 1078.01    89.8 1071.65   109.8 1067.63   149.7 1051.23   159.7 1045.26
   169.7 1038.06   179.7 1034.47   189.6 1032.84   199.6 1028.88   209.6 1027.35
   229.6 1021.41   273.1 1015.09   279.5 1014.67   285.8 1015.17   309.4 1020.34
   329.4 1021.75   339.3 1023.66   398.1 1047.59   407.9 1049.91   417.7 1054.03
   427.4    1060   437.2 1061.73   446.9  1065.7   544.5 1123.27   554.3 1127.93
#Mann= 3 , 0 , 0
       0      .1       0   273.1    .045       0   285.8      .1       0
Bank Sta=273.1,285.8
XS Rating Curve= 0 ,0
Exp/Cntr=0.3,0.1

Type RM Length L Ch R = 1 ,9201.9  ,169.1,176.1,183.1
XS GIS Cut Line= 3
     1705066.495      192930.679     1705009.237       193108.18
     1705035.003      193446.006
#Sta/Elev= 30
     9.8  1124.8    39.3 1107.24    49.1 1106.88    58.9 1101.88    78.5 1089.57
    98.2  1078.5   117.8 1068.43   147.2 1054.12   157.1 1054.36   186.5  1040.6
   206.4 1030.49   216.4 1027.72   226.4  1026.2   236.3 1023.13   246.3    1018
   259.9 1015.12   266.2 1014.24   272.6 1015.13   276.2 1015.62   286.2  1018.7
   296.1 1019.38   316.1 1018.57   375.8 1021.89   385.8 1022.84   415.7 1027.99
   465.5  1038.9   475.5  1039.7   485.5 1044.74   505.4  1057.8   525.3  1068.9
#Mann= 3 , 0 , 0
       0      .1       0   259.9    .045       0   272.6      .1       0
Bank Sta=259.9,272.6
XS Rating Curve= 0 ,0
Exp/Cntr=0.3,0.1

Type RM Length L Ch R = 1 ,9025.8  ,311.9,320.6,329.4
XS GIS Cut Line= 3
     1704920.861      192926.077     1704858.484      193140.497
      1704756.85       193515.54
#Sta/Elev= 30
     9.7 1153.99    29.1 1139.27    38.8 1134.77    48.5 1131.25    77.7 1105.11
    87.4 1096.91    97.1 1089.42   116.5 1076.03   135.9 1063.08   155.3 1056.57
   203.9 1024.25   213.6 1020.92   233.3 1020.61   253.2 1018.86   263.2 1016.36
   273.1 1011.85   276.7 1011.22   283.1 1010.11   289.5 1011.79     303 1016.58
     313 1018.58   372.8 1020.66   472.4 1027.29   492.3 1030.36   522.2 1033.96
   532.2 1036.45   552.1 1042.94   562.1 1045.09     582  1047.5   611.9 1049.22
#Mann= 3 , 0 , 0
       0      .1       0   276.7    .045       0   289.5      .1       0
Bank Sta=276.7,289.5
XS Rating Curve= 0 ,0
Exp/Cntr=0.3,0.1

Type RM Length L Ch R = 1 ,8705.1  ,318.1,325.5,333
XS GIS Cut Line= 3
     1704761.826      192813.564     1704482.009       193153.38
     1704406.141      193296.526
#Sta/Elev= 30
      10 1156.65      30 1140.68      40 1137.49      50 1132.83      70  1120.5
   120.1 1087.75   130.1 1080.52   140.1  1071.6   160.1 1057.03   180.1 1048.81
   210.1  1027.7   220.1 1022.68   240.1 1019.36   260.1 1009.66   263.7 1009.01
   270.1 1007.84   276.5 1008.46   290.1 1009.71   310.1 1013.33   350.2 1017.07
   390.2 1022.34   410.2  1029.4   430.2  1034.8   460.4 1050.07   470.6 1058.12
   511.1  1081.4   521.2 1086.28   531.3 1088.65   561.7 1109.18   602.2 1140.96
#Mann= 3 , 0 , 0
       0      .1       0   263.7    .045       0   276.5      .1       0
Bank Sta=263.7,276.5
XS Rating Curve= 0 ,0
Exp/Cntr=0.3,0.1

Type RM Length L Ch R = 1 ,8379.6  ,312.1,311.5,310.9
XS GIS Cut Line= 3
      1704564.38      192670.569     1704326.721      192803.802
     1704106.383      192970.141
#Sta/Elev= 30
    10.1 1111.34    60.5 1076.29    80.7  1056.3    90.8 1049.37     111 1039.26
   131.2 1026.47   141.3 1020.98   161.5 1013.94   171.5 1009.18   181.6 1005.81
   185.3 1005.69   191.7 1005.49   198.2 1006.87   211.9 1010.61     222 1012.53
   262.4 1018.67   272.5 1021.52   282.3 1023.13   311.9 1031.87   321.8 1036.76
   371.1  1053.6   400.6 1065.12   410.5 1069.45   420.4 1076.27   430.2 1080.61
   449.9 1084.34   479.5 1092.81   499.2  1099.8     519 1111.82   548.5 1127.46
#Mann= 3 , 0 , 0
       0      .1       0   185.3    .045       0   198.2      .1       0
Bank Sta=185.3,198.2
XS Rating Curve= 0 ,0
Exp/Cntr=0.3,0.1

Type RM Length L Ch R = 1 ,8068.1  ,343,348.7,354.5
XS GIS Cut Line= 2
      1704366.06      192420.471     1704042.549      192616.581
#Sta/Elev= 30
      10 1059.35    19.9 1053.25    29.9 1048.37    39.8 1045.04    49.8 1042.67
    59.7 1038.39    69.7 1032.49    89.6 1020.13    99.6 1014.22   109.5 1010.58
   119.5 1009.03   129.4 1006.29   139.4    1004   149.3 1002.12   152.8 1002.04
   159.3 1001.88   165.8 1003.02   169.2 1003.62   179.2 1006.45   189.2 1008.81
     219 1012.46   268.8 1017.01   278.8 1018.99   288.7 1022.86   298.7 1028.44
   308.6 1035.29   318.6  1039.5   338.5 1050.22   358.4 1061.39   378.3 1073.02
#Mann= 3 , 0 , 0
       0      .1       0   152.8    .045       0   165.8      .1       0
Bank Sta=152.8,165.8
XS Rating Curve= 0 ,0
Exp/Cntr=0.3,0.1

Type RM Length L Ch R = 1 ,7719.3  ,210.5,215,219.5
XS GIS Cut Line= 3
     1704275.878       192145.63     1703882.763      192250.455
     1703870.518      192453.846
#Sta/Elev= 30
     9.9 1072.02    39.7 1059.69    49.6 1051.75    59.5 1045.22    89.3 1030.33
    99.2 1024.31     129 1004.04   148.8 1002.82   208.4 1003.86   228.2   998.9
   231.6  998.68   238.2  998.25   244.7  999.71     258  1002.8   327.5 1006.79
   357.2 1010.96   367.2 1013.73   377.1  1015.2   406.9 1018.88   416.6 1019.02
   426.3 1020.71   484.5 1046.88   503.9 1054.44   523.3 1057.61   562.1 1067.55
   571.8 1071.24   581.5 1075.79   591.2 1081.81   600.9 1090.03   610.6 1095.28
#Mann= 3 , 0 , 0
       0     .08       0   231.6    .045       0   244.7      .1       0
Bank Sta=231.6,244.7
XS Rating Curve= 0 ,0
Exp/Cntr=0.3,0.1

Type RM Length L Ch R = 1 ,7504.3  ,361.4,365.4,369.4
XS GIS Cut Line= 4
      1704287.33      192019.661     1704194.822      191999.949
     1703861.291      192011.401      1703690.41      192031.113
#Sta/Elev= 30
     9.5 1047.97    56.8 1027.52    66.2 1022.78    75.7 1015.35    85.1 1011.21
    94.6 1008.07   114.8 1003.41   124.9  1001.8   165.4  998.99   195.7  998.02
   266.5  998.96   286.7  999.94   296.8  999.16     307  995.36   310.5  995.27
   317.1  995.09   323.6  996.85   337.3 1001.88   347.4 1004.35   408.1 1011.53
   428.3 1015.98   448.5 1021.59   458.7 1027.38   478.9 1035.92   509.3 1053.96
   519.4 1060.64   539.6    1079   549.7    1084     570 1092.32   600.3 1107.34
#Mann= 3 , 0 , 0
       0     .08       0   310.5    .045       0   323.6      .1       0
Bank Sta=310.5,323.6
XS Rating Curve= 0 ,0
Exp/Cntr=0.3,0.1

Type RM Length L Ch R = 1 ,7139    ,232.8,229.2,225.6
XS GIS Cut Line= 3
     1704330.274      191706.171     1703968.113      191650.344
      1703781.76      191617.168
#Sta/Elev= 30
     9.9 1016.41    49.5 1012.92    69.3 1008.93      99 1003.99   118.8 1001.01
   128.7  999.93   158.5  998.74   198.1  999.11   217.9  997.79   247.6  991.11
   260.8  988.94   267.4  988.37     274  988.52   287.2  989.67     307  993.87
   326.8  996.47   336.7  998.75   346.6 1003.46   366.4 1015.88   376.4 1022.83
   386.4 1032.33   416.2 1049.49   456.1 1071.22   466.1 1084.31     476 1090.35
     486 1095.55   525.8 1115.35   535.8 1125.48   545.8 1133.06   555.7 1139.27
#Mann= 3 , 0 , 0
       0      .1       0   260.8    .045       0     274      .1       0
Bank Sta=260.8,274
XS Rating Curve= 0 ,0
Exp/Cntr=0.3,0.1

Type RM Length L Ch R = 1 ,6909.8  ,302.9,298.1,293.2
XS GIS Cut Line= 2
     1704278.741      191435.624     1703802.064      191448.507
#Sta/Elev= 30
     9.9 1018.17    39.7 1005.57    49.7 1002.53    59.6 1000.53    69.5  999.68
    79.5  999.25    89.4  998.51    99.3  997.48   119.2     994     149  990.43
   178.8  986.52   182.1  986.41   188.8  986.17   195.4  986.74   248.4  992.97
   258.3  994.35   268.2   997.9   278.2  1000.9     298 1007.65     308  1011.3
   317.9 1015.26   327.8 1019.59   337.8 1024.21   347.7 1033.68   357.6 1038.74
   407.3  1062.3   417.2 1071.32   427.2 1077.34     457 1093.13   476.9 1104.22
#Mann= 3 , 0 , 0
       0      .1       0   182.1    .045       0   195.4      .1       0
Bank Sta=182.1,195.4
XS Rating Curve= 0 ,0
Exp/Cntr=0.3,0.1

Type RM Length L Ch R = 1 ,6611.7  ,321.5,314.3,307
XS GIS Cut Line= 2
     1704262.995       191089.21     1703767.099      191223.761
#Sta/Elev= 30
    10.1 1074.36    40.3 1059.97    50.4 1051.61   120.9 1021.16     131 1014.12
   141.1 1008.55   151.1 1004.61   161.2 1002.07   181.4 1000.58   191.4  998.92
   201.5  995.73   211.6  992.02   241.8   984.7   251.9  983.38   255.3  983.37
     262  983.35   268.6  984.11     272   984.5   282.1  987.42   322.4  993.24
   332.5  995.92   342.6   999.9   352.6 1004.33   362.7 1011.88   372.8 1017.39
   423.2 1040.75   443.3 1055.34   483.6 1074.57   503.8 1085.06   513.8 1091.13
#Mann= 3 , 0 , 0
       0      .1       0   255.3    .045       0   268.6      .1       0
Bank Sta=255.3,268.6
XS Rating Curve= 0 ,0
Exp/Cntr=0.3,0.1

Type RM Length L Ch R = 1 ,6297.4  ,289.1,278.7,268.4
XS GIS Cut Line= 3
     1704102.671      190715.598     1703746.774      190970.727
     1703633.004      191004.158
#Sta/Elev= 30
      10 1049.22    19.9 1047.52    39.8  1040.1    49.8 1038.07    69.7 1034.88
    89.6  1029.8    99.5 1027.63   159.2 1015.64   218.9 1002.94   238.9  1000.5
   248.8  997.56   258.8  987.03   268.7  981.42     272  981.09   278.7  980.41
   285.4  980.56   288.6  980.64   348.3  986.71   358.3  988.37   378.2  990.82
   388.1   992.8   398.1  996.75   427.9 1011.83   437.9 1017.48   447.8 1025.15
   477.4 1039.51   507.1 1054.86     517 1062.48   536.7 1069.61   556.5 1080.33
#Mann= 3 , 0 , 0
       0      .1       0     272    .045       0   285.4      .1       0
Bank Sta=272,285.4
XS Rating Curve= 0 ,0
Exp/Cntr=0.3,0.1

Type RM Length L Ch R = 1 ,6018.7  ,312.1,321.9,331.7
XS GIS Cut Line= 3
      1703769.14      190479.407     1703624.562      190791.466
     1703499.931      190948.373
#Sta/Elev= 30
    10.1  1038.5    30.3 1035.62    60.7 1032.96    70.8 1030.49   101.2 1020.21
   121.4 1016.03   141.6 1006.74   161.8  999.28     172  996.69   192.2  994.61
   202.3  992.57   222.5   985.3   232.7  984.01     236  982.73   242.8   980.1
   249.5  981.76     263  987.44   273.1  988.54   303.5  988.89   353.9  991.56
     364  992.67     374  996.69     404 1018.39   424.1 1036.19   444.1 1050.38
   454.1 1053.38   464.2 1058.36   514.2 1094.71   534.3 1110.69   544.3 1117.32
#Mann= 3 , 0 , 0
       0      .1       0     236    .045       0   249.5      .1       0
Bank Sta=236,249.5
XS Rating Curve= 0 ,0
Exp/Cntr=0.3,0.1

Type RM Length L Ch R = 1 ,5696.8  ,353.2,344.3,335.8
XS GIS Cut Line= 4
     1703568.244      190323.357     1703494.299      190508.036
     1703249.519      190694.126     1703180.809      190810.075
#Sta/Elev= 30
     9.9 1038.97    29.8 1033.85    49.7  1030.6    59.7  1027.6    69.6 1023.29
    79.6 1017.59    89.5  1010.7    99.5 1005.13   109.4 1001.28   119.4  998.46
   139.3  994.24   159.1  992.61     189  988.52   298.1  981.84   340.9  978.17
   347.7  977.54   354.5  977.61   357.6  977.64   367.6  979.41   407.2  990.18
   427.1  994.82   446.9  997.86   466.7 1004.34   476.7 1008.31   496.5 1017.52
   554.6 1035.96   573.8 1037.74   602.7 1045.25   621.9 1048.92   641.2  1053.7
#Mann= 3 , 0 , 0
       0     .08       0   340.9    .045       0   354.5      .1       0
Bank Sta=340.9,354.5
XS Rating Curve= 0 ,0
Exp/Cntr=0.3,0.1

Type RM Length L Ch R = 1 ,5352.5  ,37.6,37.5,37.3
XS GIS Cut Line= 3
     1703459.676      190200.271     1703251.398      190292.601
     1703078.548      190591.061
#Sta/Elev= 30
     9.9 1045.18    19.8 1038.68    29.7 1034.12    49.5 1025.97    79.2  1016.4
    89.1 1012.79    99.1 1010.05     109 1009.13   158.5  997.76   168.4  995.07
   178.3  993.35   227.8  987.99   257.4  983.38   277.1  979.73     287   975.1
     290  974.74   296.8  973.93   303.6  974.99   326.4  979.39   355.9   982.2
   454.5  982.69   464.3  983.16   474.2  986.09   493.9  997.21   513.6 1003.71
   523.5 1009.57   533.3 1016.48   543.2 1025.87     553 1033.81   572.7 1042.39
#Mann= 3 , 0 , 0
     9.9      .1       0     290    .045       0   303.6      .1       0
#XS Ineff= 2 , 0
       0     282             317       0
Permanent Ineff=
       F       F
Bank Sta=290,303.6
XS Rating Curve= 0 ,0
Exp/Cntr=0.3,0.1

Type RM Length L Ch R = 1 ,5315.1  ,204.8,208.6,212.3
XS GIS Cut Line= 3
       1703287.9      190066.072      1703234.22      190246.436
      1703046.34      190574.957
#Sta/Elev= 30
     9.9 1086.39    19.8  1075.3    29.7 1065.18    49.5 1047.03    59.4 1040.52
    69.3 1039.22    89.1 1025.34   108.9  1014.3   118.9 1009.66   138.7 1002.16
   158.5  996.58   178.3  994.46     228  985.19   247.9  983.24   257.9  981.32
   277.8  973.91   280.9  973.75   287.8  973.42   294.6  973.69   327.6  980.01
   347.5  981.65   437.2  982.23   457.1  983.35     467  987.99     477  995.18
   496.9 1007.38   506.9 1012.42   516.8 1014.91   536.8 1026.08   566.6 1041.46
#Mann= 3 , 0 , 0
     9.9      .1       0   280.9    .045       0   294.6      .1       0
#XS Ineff= 2 , 0
       0     278             300       0
Permanent Ineff=
       F       F
Bank Sta=280.9,294.6
XS Rating Curve= 0 ,0
Exp/Cntr=0.3,0.1

Type RM Length L Ch R = 1 ,5106.5  ,378.9,366.9,354.9
XS GIS Cut Line= 3
     1703186.549      190019.843     1702903.552      190348.428
      1702825.59      190437.877
#Sta/Elev= 30
    10.1 1104.65    80.7 1060.32    90.8 1053.45   100.8 1047.53     121 1036.53
   131.1 1036.22   141.2 1031.44   161.4 1019.85   181.5 1007.67   191.6 1000.33
   201.7  993.71   211.8  988.56     232  984.77     242  982.03   252.1  980.74
   272.3  971.64   275.5  970.96   282.4  969.51   289.2  969.76   373.1  979.11
   393.3  980.06   423.6  983.16   433.7  985.31   443.5  988.43   463.3  995.89
     493 1008.41   502.9 1009.91   512.8 1012.81   522.6 1017.81   552.3 1030.94
#Mann= 3 , 0 , 0
       0      .1       0   275.5    .045       0   289.2      .1       0
Bank Sta=275.5,289.2
XS Rating Curve= 0 ,0
Exp/Cntr=0.3,0.1

Type RM Length L Ch R = 1 ,4739.6  ,295.1,311.1,327.1
XS GIS Cut Line= 4
     1702769.714      189848.517      1702679.17      190033.864
     1702658.772       190208.86     1702470.158      190323.756
#Sta/Elev= 30
     9.8 1060.44    19.6 1055.58    39.3 1049.55    49.1 1045.29    58.9 1040.78
    78.6 1029.83    88.4 1025.86   127.7 1010.68   147.3 1005.74   196.5  986.71
   206.3  983.78   225.9  982.31   255.2  978.39     265  975.69   277.7   970.2
   284.6  967.88   291.5  968.45   294.4  968.69   304.2  972.88   313.9  975.56
   353.1   976.9   392.5  981.25   422.6  982.36   432.7   985.4   452.7 1002.83
   462.8 1008.98   472.8 1012.99   492.9 1016.99     513    1019   603.3 1051.44
#Mann= 3 , 0 , 0
       0      .1       0   277.7    .045       0   291.5      .1       0
Bank Sta=277.7,291.5
XS Rating Curve= 0 ,0
Exp/Cntr=0.3,0.1
